--- PIPESTCK.prj (project) ---

Proj Title=PIPESTCK
Current Plan=p01
Default Exp/Contr=0,0
English Units
Geom File=g01
Flow File=f01
Plan File=p01
BEGIN DESCRIPTION:
END DESCRIPTION:
DSS Export Rating Curves= 0
DSS Export Rating Curve Sorted= 0
DSS Export Volume Flow Curves= 0
DXF OffsetX= 0
DXF OffsetY= 0
DXF ScaleX= 0
DXF ScaleY= 0

--- PIPESTCK.p01 (plan) ---

Plan Title=Floodplain
Program Version=4.00
Geom File=g01
Flow File=f01
K Sum by GR=0
Std Step Tol=0.01
Critical Tol=0.01
Num of Std Step Trials=20
Max Error Tol=0.3
Flow Tol Ratio=0.001
Split Flow NTrial=30
Split Flow Tol=0.02
Split Flow Ratio=0.02
Log Output Level=0
Friction Slope Method=1
Unsteady Friction Slope Method=2
Unsteady Bridges Friction Slope Method=1
Global Log Level=0
CheckData=False
Run HTab=0
Run UNet=0
Run PostProcess=0
UNET Theta=0
UNET Theta Warmup=0
UNET ZTol=0
UNET ZSATol=0
UNET MxIter=0
UNET MaxInSteps=0
UNET DtIC=0
UNET DtMin=0
UNET MaxCRTS=0
UNET WFStab=0
UNET SFStab=0
UNET WFX=0
UNET SFX=0
UNET DSS MLevel=0
UNET DZMax Abort=0
UNET Convert EG Bridges=0
UNET Use Existing IB Tables=0
UNET Froude Limit=0
UNET Froude Power=0
Write IC File=0
Echo Input=False
Echo Output=False
Write Detailed=0

--- PIPESTCK.f01 (steady flow) ---

Flow Title=2010 USGS WV Regression Equation
Program Version=5.03
Number of Profiles= 1
Profile Names=P100yr
River Rch & RM=PIPESTCK,Main            ,27169.9
505.2999
River Rch & RM=PIPESTCK,Main            ,26720.8
505.3746
River Rch & RM=PIPESTCK,Main            ,26276.2
717.2589
River Rch & RM=PIPESTCK,Main            ,24801.4
780.3663
River Rch & RM=PIPESTCK,Main            ,23132
829.7194
River Rch & RM=PIPESTCK,Main            ,20918.7
895.2061
River Rch & RM=PIPESTCK,Main            ,15911
983.1546
River Rch & RM=PIPESTCK,Main            ,14870.9
1152.223
River Rch & RM=PIPESTCK,Main            ,12711.1
1228.424
River Rch & RM=PIPESTCK,Main            ,7361.4
1345.861
River Rch & RM=PIPESTCK,Main            ,7066.5
 1672.66
River Rch & RM=PIPESTCK,Main            ,6180.6
1702.524
River Rch & RM=PIPESTCK,Main            ,4372.9
1881.393
River Rch & RM=PIPESTCK,Main            ,150.3
2016.862
Boundary for River Rch & Prof#=PIPESTCK,Main            , 1
Up Type= 0
Dn Type= 1
Dn Known WS=1684.5
DSS Import GetInterval= 0
DSS Import GetPeak= 0
DSS Import FillOption= 0

--- PIPESTCK.g01 (geometry) ---

Geom Title=LiDAR
Program Version=4.10

River Reach=PIPESTCK        ,Main
Reach XY= 30
     1978324.091      193959.454      1978250.48      194132.718
     1978439.021       194233.76     1978656.035      194817.093
     1978607.654      195165.358     1979066.749      195437.033
     1979234.616      195756.025     1979206.491      196566.442
     1979484.095      196794.567     1979517.158      197546.772
     1979655.159      197548.209     1979995.232       198273.76
     1980475.319      198354.837     1981087.224       198727.37
     1980681.495      199222.683     1980207.133      199216.816
      1980322.12      199743.516     1980603.077      200072.382
     1981591.786      200420.219     1982161.703      201341.954
     1983262.745      202079.454     1983754.411       202701.85
     1984174.724      202904.454     1985727.849      203162.266
     1987752.328      204444.037     1989374.724      204913.829
     1990899.909       206358.69     1992555.924      207456.078
     1992809.326       207987.45     1994076.764      209104.711

Type RM Length L Ch R = 1 ,27169.9 ,462,449,427.7
XS GIS Cut Line= 3
     1977849.304      193701.855     1978396.179      194040.397
     1978713.019      194014.355
#Sta/Elev= 30
       0 2399.58    71.8 2398.99    94.7 2397.18   104.5 2398.88   150.2 2399.02
   199.2 2398.69   212.2 2397.68     271 2398.69   313.4  2397.4     333 2398.28
   408.1    2397   515.8 2397.96   522.4 2397.47   528.9 2395.31   535.4 2393.22
   538.7 2393.04  543.242395.489   545.2 2396.91   548.5  2397.3  574.812396.637
   607.3  2398.7   656.3 2397.51     676 2398.73   682.5  2398.2   708.7 2400.44
   748.1 2402.55   816.9 2404.66   902.1 2410.58   934.9 2410.49   961.1 2411.52
#Mann= 4 ,-1 , 0
       0     .08       0   528.9    .045       0  543.24     .08       0
  574.81     .12       0
#XS Ineff= 2 , 0
          331.27 2399.92  614.04         2399.63
Permanent Ineff=
       F       F
Bank Sta=528.9,543.24
XS Rating Curve= 0 ,0
Exp/Cntr=0.3,0.1

Type RM Length L Ch R = 1 ,26720.8 ,185.8,177.5,149.2
XS GIS Cut Line= 3
     1977815.428      194285.297     1978586.261      194256.651
     1978742.511       194212.38
#Sta/Elev= 30
       0 2403.71      36 2401.82   46.652401.889    91.5 2398.83   143.8 2397.79
   228.8 2397.83   369.3  2396.9   424.9 2397.51   496.8 2396.98  538.632397.356
   558.9 2396.29   585.1 2396.17   594.9 2395.47   611.2 2396.24  616.582394.814
     621 2393.07   627.6 2393.72  632.072394.916   637.4 2396.54   660.2 2395.58
   686.4 2396.68   745.2 2403.48   771.4 2405.86   810.3  2408.6  818.762408.709
  849.46 2409.97   868.8 2410.34   878.6  2409.9  896.712410.056   933.8 2409.86
#Mann= 8 ,-1 , 0
       0     .12       0   46.65     .08       0  538.63     .12       0
  616.58    .045       0  632.07     .12       0  818.76     .06       0
  849.46    .016       0  896.71     .12       0
#XS Ineff= 2 , 0
          532.51 2397.84
Permanent Ineff=
       F       F
Bank Sta=616.58,632.07
XS Rating Curve= 0 ,0
Exp/Cntr=0.3,0.1

Type RM Length L Ch R = 1 ,26543.4 ,27.9,26.5,26.7
XS GIS Cut Line= 2
      1977909.59      194724.867     1978737.586      194257.186
#Sta/Elev= 30
       0 2416.86    16.4 2416.07   36.632414.065   97.672406.648   127.9 2399.45
   167.2 2397.14   367.3 2395.66   377.1 2396.11   406.6 2395.78     446 2396.24
   590.2 2395.93   613.2 2394.75   655.8 2395.22   662.4 2394.24   665.7 2392.36
   668.9 2390.99   675.5 2391.48   678.8 2392.55   685.3 2394.97   688.6 2395.55
   714.8 2397.22   760.8 2402.38   803.4  2406.2   836.2 2407.76   859.1  2407.8
   885.4 2409.17  893.392408.891   918.2 2409.16   937.8 2408.49     951 2409.02
#Mann= 6 ,-1 , 0
       0     .06       0   36.63     .12       0   97.67    .016       0
   665.7    .045       0   678.8    .016       0  893.39     .12       0
#XS Ineff= 2 , 0
           538.7  2397.3
Permanent Ineff=
       F       F
Bank Sta=665.7,678.8
XS Rating Curve= 0 ,0
Exp/Cntr=0.3,0.1

Type RM Length L Ch R = 1 ,26516.9 ,234.5,240.6,244
XS GIS Cut Line= 2
     1977919.138      194749.172     1978747.135      194281.491
#Sta/Elev= 30
       0 2417.46   37.862414.538   62.542412.072    65.6 2411.71    88.5 2405.41
   108.2 2401.77   121.3 2400.98   134.4 2399.36   154.1 2398.48   216.4 2396.81
   324.6 2396.18   485.3 2396.19   573.8 2395.61   590.2    2396   603.4 2395.37
   629.6 2396.38   655.8 2394.78   661.7 2392.93   668.9 2390.79   672.2  2391.1
   676.7  2393.1   682.1 2395.89   698.5 2395.98     728 2397.55  772.212401.646
  804.172404.409   832.9 2405.88  870.66 2406.51   901.8 2406.84     951 2408.35
#Mann= 8 ,-1 , 0
       0     .06       0   37.86     .12       0   62.54    .016       0
   661.7    .045       0   676.7    .016       0  772.21     .12       0
  804.17    .016       0  870.66     .12       0
#XS Ineff= 2 , 0
          486.07 2396.84
Permanent Ineff=
       F       F
Bank Sta=661.7,676.7
XS Rating Curve= 0 ,0
Exp/Cntr=0.3,0.1

Type RM Length L Ch R = 1 ,26276.2 ,286.2,278.2,263.8
XS GIS Cut Line= 3
     1978052.407      194892.068     1978146.157      194780.089
     1978820.636      194527.484
#Sta/Elev= 30
       0 2420.11    42.2 2417.96    64.9 2415.71    74.6 2413.91   120.1 2401.18
   136.3 2397.28  157.882396.089   260.6 2394.94   434.1 2395.36   489.8 2395.02
   506.2 2394.36   574.9 2395.03   581.4 2394.42  585.682392.435     588 2391.05
   594.6 2390.17  600.182392.636   604.4 2394.26   620.7 2394.06   637.1 2395.71
  654.47 2396.18   666.6 2396.16   682.9 2394.93   702.6 2394.31     732 2394.23
   758.2 2396.16   787.7 2399.59   794.2 2399.64   830.3 2402.86   866.3 2404.46
#Mann= 5 ,-1 , 0
       0     .12       0  157.88     .08       0  585.68    .045       0
  600.18     .08       0  654.47     .12       0
#XS Ineff= 2 , 0
          433.44  2396.5  651.19         2397.04
Permanent Ineff=
       F       F
Bank Sta=585.68,600.18
XS Rating Curve= 0 ,0
Exp/Cntr=0.3,0.1

Type RM Length L Ch R = 1 ,25998   ,470.2,492.1,490.8
XS GIS Cut Line= 3
     1978255.573       195168.11     1978713.907      194712.381
     1978875.365      194631.652
#Sta/Elev= 30
       0 2422.86    32.6 2423.11    78.3 2422.67     111 2421.08   127.3  2418.6
   169.8 2406.35   182.8 2401.89   195.9  2398.4   212.2 2395.36   218.7 2394.75
   277.5 2394.42     346  2392.8   375.4 2393.45   411.3 2392.98     457 2393.11
   522.3 2394.67   528.8 2394.13   535.4 2392.13   538.6 2390.87   541.9 2390.68
  549.812392.189   554.9 2393.25     568 2393.15   590.8 2395.46     685 2395.34
   710.8 2397.49   749.5 2402.34   768.8 2402.75   781.7  2404.2   826.9 2407.42
#Mann= 3 , 0 , 0
       0     .12       0   535.4    .045       0  549.81     .12       0
#XS Ineff= 2 , 0
          378.74  2396.5   590.3         2396.39
Permanent Ineff=
       F       F
Bank Sta=535.4,549.81
XS Rating Curve= 0 ,0
Exp/Cntr=0.3,0.1

Type RM Length L Ch R = 1 ,25506   ,713.1,704.6,694.3
XS GIS Cut Line= 2
     1978351.886      195358.214     1979052.407      194855.609
#Sta/Elev= 30
       0  2411.1    65.6 2414.94   111.5  2416.2   144.2 2415.74   196.7  2413.1
   222.9 2410.91   262.3 2406.02   285.2 2402.67     295 2400.66   301.6 2398.61
   304.9 2396.42  309.772392.294   311.4 2391.01   314.7 2389.45   321.3 2389.04
   324.5 2389.49   327.8 2391.36   331.1 2392.35  339.76 2392.61   350.8 2392.18
   383.6 2392.24   396.7 2393.04  443.862392.365     518 2393.26   665.5 2392.74
  694.172393.442   711.4 2394.18  764.842399.528   826.1 2405.66   862.2 2408.36
#Mann= 7 ,-1 , 0
       0     .12       0  309.77    .045       0   331.1     .12       0
  339.76     .08       0  443.86     .06       0  694.17     .12       0
  764.84     .06       0
#XS Ineff= 2 , 0
                          518.06         2394.99
Permanent Ineff=
       F       F
Bank Sta=309.77,331.1
XS Rating Curve= 0 ,0
Exp/Cntr=0.3,0.1

Type RM Length L Ch R = 1 ,24801.4 ,755.7,766.5,772.8
XS GIS Cut Line= 2
     1978588.866      195764.464     1979422.199      195355.609
#Sta/Elev= 30
       0 2417.24      59 2416.52   114.8 2412.26   209.9 2402.55   236.2 2401.67
  314.992397.735   334.6 2396.98  348.312395.534   360.8 2395.34     410 2392.08
   465.8 2391.32     492 2389.18   524.8 2389.28   541.2  2390.5   544.5 2390.42
  549.362389.196   554.3 2387.82   564.2 2389.18   570.7 2390.44   590.4 2390.12
   659.3 2390.87   692.1 2391.72   744.6 2392.23   770.8 2393.09   826.6    2400
   875.8 2403.88   892.2 2404.22   902.32405.626  917.092407.011   928.2 2407.61
#Mann= 7 ,-1 , 0
       0     .06       0  314.99     .12       0  348.31     .08       0
  549.36    .045       0   564.2     .08       0   902.3     .12       0
  917.09    .016       0
Bank Sta=549.36,564.2
XS Rating Curve= 0 ,0
Exp/Cntr=0.3,0.1

Type RM Length L Ch R = 1 ,24034.9 ,818.2,902.8,827.3
XS GIS Cut Line= 2
     1978765.949      196235.818     1979573.241      196173.318
#Sta/Elev= 30
       0 2403.72     6.6 2404.28     9.8 2403.79   17.942400.343    29.5 2394.63
   37.632393.212      59 2393.08    72.1 2391.37   275.4 2387.95   327.8 2388.35
   367.2 2387.12   386.8 2387.97   422.9  2386.2     436 2387.71   472.1  2387.5
   511.4  2388.4   514.7 2388.15  518.812386.476   521.2 2385.05   527.8 2384.56
   531.1 2384.98   534.3 2386.51   537.6 2388.05   540.9 2388.28     554 2388.08
   593.4 2390.73  688.942393.735   770.4 2395.44   786.8 2397.52   809.7 2397.55
#Mann= 6 ,-1 , 0
       0     .04       0   17.94     .12       0   37.63     .08       0
  518.81    .045       0   534.3     .08       0  688.94     .12       0
Bank Sta=518.81,534.3
XS Rating Curve= 0 ,0
Exp/Cntr=0.3,0.1

Type RM Length L Ch R = 1 ,23132   ,1300.3,1348.9,1065.6
XS GIS Cut Line= 2
     1978768.553      197011.859     1979755.532       196649.88
#Sta/Elev= 30
       0 2398.48    29.5 2400.44    52.4 2400.49    65.5 2398.85    98.2 2392.12
   121.2  2389.1   248.52386.629   271.8 2385.17   288.2  2387.6     298 2387.86
  320.792386.294  393.612386.233  433.772386.229   566.6 2386.74  608.762385.641
   661.5    2385   707.4 2385.28   717.2 2386.08     727 2384.56   736.9 2384.24
  740.952384.567   756.5 2385.46   779.4 2388.73  839.462393.431   903.9 2396.72
   956.3 2401.26  1010.72404.685  1041.4  2404.3  1045.52405.121  1051.3  2407.1
#Mann= 11 ,-1 , 0
       0     .12       0   248.5     .06       0  320.79     .12       0
  393.61     .06       0  433.77     .12       0  608.76     .08       0
     727    .045       0  740.95     .08       0  839.46     .12       0
  1010.7    .016       0  1045.5     .12       0
#XS Ineff= 2 , 0
          294.74 2388.72
Permanent Ineff=
       F       F
Bank Sta=727,740.95
XS Rating Curve= 0 ,0
Exp/Cntr=0.3,0.1

Type RM Length L Ch R = 1 ,21783.2 ,448.4,452.5,449.8
XS GIS Cut Line= 2
     1979134.438      197781.521     1980002.494      197392.632
#Sta/Elev= 30
       0 2413.21    72.2 2417.76   127.9 2419.59   177.1 2419.95   196.8 2419.14
   252.6 2413.48     305 2405.22   324.7 2400.39   357.5    2388   367.4 2385.24
   400.2    2383  444.912383.393   505.1 2382.92   521.5 2381.91   541.2 2382.49
   564.2 2381.11   570.7  2380.2   580.6 2381.19  614.512382.774   649.4 2383.26
   692.1 2385.56   741.3 2385.63     797 2386.93  813.45 2388.61  841.082393.015
   859.4 2392.91  868.092392.085     879 2394.29   931.5 2396.92   951.2 2399.12
#Mann= 8 ,-1 , 0
       0     .06       0  444.91     .07       0   564.2    .045       0
   580.6     .07       0  614.51     .06       0  813.45     .08       0
  841.08    .016       0  868.09     .12       0
Bank Sta=564.2,580.6
XS Rating Curve= 0 ,0
Exp/Cntr=0.3,0.1

Type RM Length L Ch R = 1 ,21330.7 ,218.8,211.7,202.6
XS GIS Cut Line= 2
     1979440.862      198083.604     1980024.195      197847.493
#Sta/Elev= 30
       0 2387.99    75.4 2386.18   121.3 2384.79   134.4 2384.58   144.2 2384.74
     177 2383.46   196.7 2383.21   199.9 2383.37   245.8 2382.59   265.5 2382.57
   314.6  2381.3     331 2381.11  341.822380.427   350.7 2379.27   360.5  2378.6
   363.8 2378.72   367.1 2379.31   370.4 2379.84   376.9 2379.65   386.8 2380.96
   393.3  2381.5   419.5 2382.19   504.8  2385.1     531 2386.73   540.8 2387.67
   557.2 2388.23   563.8 2388.68  582.722388.652   599.8 2389.61   629.3 2390.63
#Mann= 5 ,-1 , 0
       0     .06       0  341.82     .12       0   350.7    .045       0
   367.1     .06       0  582.72    .016       0
Bank Sta=350.7,367.1
XS Rating Curve= 0 ,0
Exp/Cntr=0.3,0.1

Type RM Length L Ch R = 1 ,21119   ,221.5,200.3,176.8
XS GIS Cut Line= 3
     1979631.545      198353.208     1979953.811      198060.239
     1980091.614      198010.326
#Sta/Elev= 30
       0 2384.62    78.6 2383.46   134.3 2382.35   186.7 2380.91   212.8 2381.18
   222.7 2380.77   235.8 2380.76     239 2380.43   245.6 2380.88   252.2 2380.55
     262  2380.9   268.5  2380.4   294.7 2379.66   325.62379.412   332.3 2378.57
   337.3 2377.63   340.6 2377.55  346.122378.598   350.4 2379.48   360.2 2380.53
   383.1 2381.03   406.1 2382.51  437.982383.818   448.6 2383.87  474.692385.172
   490.9 2386.84   506.12387.437   523.5  2387.6  537.522388.644   582.1 2391.84
#Mann= 8 ,-1 , 0
       0     .06       0   325.6     .12       0   332.3    .045       0
  346.12     .06       0  437.98     .12       0  474.69    .016       0
   506.1     .06       0  537.52     .12       0
#XS Ineff= 2 , 0
           79.26 2384.46
Permanent Ineff=
       F       F
Bank Sta=332.3,346.12
XS Rating Curve= 0 ,0
Exp/Cntr=0.3,0.1

Type RM Length L Ch R = 1 ,20918.7 ,56.2,56.2,55.8
XS GIS Cut Line= 4
     1979850.729      198569.137     1980009.149      198302.209
     1979996.186      198142.523      1980105.72      198029.857
#Sta/Elev= 30
       0  2407.2      49 2400.64      98  2395.4     147 2392.26   156.8 2389.93
   173.2 2390.59   192.8  2389.2  203.44 2387.46   225.4 2384.98  237.792384.974
  306.492385.041   313.7 2384.87   316.9 2383.61   323.5 2378.91   326.8  2377.5
   333.3 2376.56   339.8  2376.9   343.1 2377.71   352.9 2383.07   359.4 2385.19
   375.8 2385.93  395.932385.738   421.6 2383.35   455.22383.326   470.6 2383.76
  490.39 2386.16  526.66 2387.21   542.6 2387.21   565.6 2388.88   627.7 2391.97
#Mann= 10 ,-1 , 0
       0     .12       0  203.44     .06       0  237.79    .016       0
  306.49     .08       0   326.8    .045       0   343.1     .08       0
  395.93     .12       0   455.2     .08       0  490.39    .016       0
  526.66     .12       0
#XS Ineff= 2 , 0
                          378.53         2387.06
Permanent Ineff=
       F       F
Bank Sta=326.8,343.1
XS Rating Curve= 0 ,0
Exp/Cntr=0.3,0.1

Type RM Length L Ch R = 1 ,20862.5 ,145.8,147.6,149.3
XS GIS Cut Line= 4
     1979904.982      198572.392     1980063.403      198305.465
     1980051.686      198161.133     1980127.422      198060.239
#Sta/Elev= 30
       0 2403.97    78.4  2396.1    94.8  2393.2   114.4 2393.33   140.5 2391.36
  154.922388.969  156.95 2388.42   163.4 2385.99   173.2 2378.86   176.4 2378.24
   192.8 2378.64  207.222381.889   212.4 2383.54  225.682384.599   251.6 2385.43
  277.782384.997   303.9 2384.34   316.8 2380.98  325.612377.569   332.9 2376.26
  341.492377.695     349 2380.49   374.8 2384.69   384.4 2385.24   432.7 2383.62
   461.7 2384.77   484.3 2387.64  515.392388.478   559.12390.443   581.4 2391.59
#Mann= 10 ,-1 , 0
       0     .12       0  154.92     .06       0  156.95     .12       0
  207.22     .06       0  225.68    .016       0  277.78     .12       0
  325.61    .045       0  341.49     .12       0  515.39     .06       0
   559.1     .12       0
#XS Ineff= 2 , 0
          254.49 2386.66
Permanent Ineff=
       F       F
Bank Sta=325.61,341.49
XS Rating Curve= 0 ,0
Exp/Cntr=0.3,0.1

Type RM Length L Ch R = 1 ,20714.8 ,219.8,223.5,226.1
XS GIS Cut Line= 2
     1980219.653      198589.753     1980199.036      198089.536
#Sta/Elev= 30
       0 2387.89    26.2 2386.16    81.8 2384.44   104.7 2382.98   160.3 2381.26
   176.7 2380.99   199.6 2379.82   209.4 2378.69   212.7 2378.56   222.5 2379.16
   238.9 2378.84     252 2379.31   261.8 2378.84   274.9 2379.45     288 2378.58
   297.8 2376.24  302.742375.739   314.1  2375.3  318.79 2375.73   320.7 2376.09
   330.5 2379.22  334.182380.021   353.4 2381.62   376.3 2382.61  384.812383.377
   402.5  2384.4   422.1 2384.77     445 2385.66   471.2 2387.78   500.6 2389.32
#Mann= 5 ,-1 , 0
       0     .12       0  302.74    .045       0  318.79     .12       0
  334.18     .06       0  384.81     .12       0
Bank Sta=302.74,318.79
XS Rating Curve= 0 ,0
Exp/Cntr=0.3,0.1

Type RM Length L Ch R = 1 ,20491.4 ,225.3,231.8,237
XS GIS Cut Line= 3
     1980409.612      198505.986     1980404.404      198403.555
     1980421.765      198222.999
#Sta/Elev= 30
       0 2396.37     9.6 2393.85    19.2 2390.86    38.5 2386.84    48.1 2384.28
    57.7 2381.92    73.7 2378.84    83.3 2377.56    86.5 2377.33   102.6 2377.53
     109 2377.31   118.8 2376.36   125.2 2375.45   138.2 2374.78   144.72373.893
   147.9 2373.79  160.822373.899   164.1 2373.98   170.6 2374.74   180.3 2375.26
   183.5 2375.68   193.3 2377.88   196.5 2378.42   212.7  2379.4   219.2 2379.95
   235.4 2380.59   251.6 2382.12   264.5 2382.57     271 2383.09     284  2383.7
#Mann= 3 ,-1 , 0
       0     .12       0   144.7    .045       0  160.82     .12       0
Bank Sta=144.7,160.82
XS Rating Curve= 0 ,0
Exp/Cntr=0.3,0.1

Type RM Length L Ch R = 1 ,20259.6 ,184.3,189.6,193.3
XS GIS Cut Line= 2
     1980550.237      198540.708     1980626.626      198323.694
#Sta/Elev= 30
       0 2397.09    16.2 2392.74    19.4 2391.63    25.9 2388.79    35.6 2385.23
    38.9 2383.82    42.1 2382.02    51.8 2375.54      68 2365.67    71.3 2364.26
    74.5 2363.89    77.8 2364.15    84.2 2365.47      94 2366.82   113.4 2369.05
   123.1 2370.75   132.8 2371.33   155.5 2371.59     162 2371.01   168.5 2372.13
   171.7 2372.03   181.5 2370.48   184.7 2370.27   197.7 2370.79   204.1 2370.71
   207.4 2371.01   217.1 2372.94   220.3  2374.2   226.8 2377.34   230.1  2378.5
#Mann= 3 ,-1 , 0
       0     .12       0      68    .045       0    84.2     .12       0
Bank Sta=68,84.2
XS Rating Curve= 0 ,0
Exp/Cntr=0.3,0.1

Type RM Length L Ch R = 1 ,20070   ,235.3,238.3,238.6
XS GIS Cut Line= 2
     1980692.598      198622.305     1980841.904      198372.305
#Sta/Elev= 30
       0 2394.42     6.5  2389.7    16.4 2384.46    19.6 2382.29    22.9 2380.56
    42.5 2372.93    55.6 2368.83    75.2 2364.25    85.1 2360.72    91.6 2359.27
   101.4 2358.49     108 2358.24   114.5 2358.45   121.1 2359.11   134.1 2361.86
   137.4 2362.17   160.3 2360.79   183.2 2361.84   199.6 2364.66   206.1 2364.57
   219.2 2367.15   222.5 2367.37     229 2366.73   235.6 2364.92   248.7 2365.52
   251.9 2366.34   261.7 2370.37   274.8 2377.73   287.9 2384.17   291.2 2386.69
#Mann= 3 ,-1 , 0
       0     .12       0   101.4    .045       0   114.5     .12       0
#XS Ineff= 2 , 0
                          140.56         2364.59
Permanent Ineff=
       F       F
Bank Sta=101.4,114.5
XS Rating Curve= 0 ,0
Exp/Cntr=0.3,0.1

Type RM Length L Ch R = 1 ,19831.7 ,309.8,340.2,366.8
XS GIS Cut Line= 2
     1980850.584      198769.874     1981069.334      198462.583
#Sta/Elev= 30
       0 2390.87     6.6 2388.18     9.8 2386.04    16.4 2380.54    26.2 2375.46
    52.5 2363.64    62.3 2360.27    68.9 2359.74   118.1 2359.48   131.2    2360
   137.8 2359.37   150.9 2357.01     164 2357.11   177.1 2356.29     187 2356.62
   190.2 2356.33   195.8 2354.47   200.1 2353.87   210.8 2354.49   219.8 2356.21
     223 2357.88   236.2    2368   262.4 2385.66   288.6  2401.1   308.3 2410.81
   311.6 2412.85   318.2 2418.82   321.4 2420.65   367.4 2430.94   377.2 2432.52
#Mann= 3 ,-1 , 0
       0     .12       0   195.8    .045       0   210.8     .12       0
Bank Sta=195.8,210.8
XS Rating Curve= 0 ,0
Exp/Cntr=0.3,0.1

Type RM Length L Ch R = 1 ,19491.5 ,219.2,240.1,260.1
XS GIS Cut Line= 2
      1980883.57      198811.541     1981211.695       198887.93
#Sta/Elev= 30
       0 2388.59    13.1 2384.33    26.2 2380.98      36 2376.71    55.6  2370.7
    62.2 2367.73      72 2364.31    78.5  2361.6      85    2360    91.6 2358.88
   101.4 2358.28   107.9 2357.47   114.5 2356.06     121 2353.15   124.3 2352.18
   127.6 2352.15   137.4    2353   143.9 2353.58   163.5 2354.05   170.1 2355.53
     193 2358.79   196.2    2359   209.3 2359.16   232.2 2355.72   261.7 2355.88
   274.8 2356.83   297.6 2359.78   317.3 2360.23   323.8 2360.71   336.9 2360.86
#Mann= 3 ,-1 , 0
       0     .12       0     121    .045       0   137.4     .12       0
#XS Ineff= 2 , 0
                          202.99         2360.74
Permanent Ineff=
       F       F
Bank Sta=121,137.4
XS Rating Curve= 0 ,0
Exp/Cntr=0.3,0.1

Type RM Length L Ch R = 1 ,19251.5 ,186.7,184.9,182.2
XS GIS Cut Line= 2
     1980871.418      198920.916     1981010.307      199207.374
#Sta/Elev= 30
       0 2377.73     6.5 2374.28    16.2 2367.52      26 2364.94    35.7 2360.71
    42.2 2359.04    48.7 2358.21    74.7 2357.12   100.7    2358   107.2  2357.8
     117  2355.9   126.7 2351.34   132.1 2350.79   139.7 2350.72   147.1 2351.03
   152.7 2351.88   155.9 2354.21   162.4 2360.53   165.7 2363.18   175.4 2368.89
   185.2 2372.65   194.9 2377.49   204.7  2381.1   237.1 2394.46   253.4 2402.99
   269.6 2407.73   285.9 2411.42   295.6 2415.21   298.9 2416.05   318.4  2417.8
#Mann= 3 ,-1 , 0
       0     .12       0   132.1    .045       0   147.1     .12       0
Bank Sta=132.1,147.1
XS Rating Curve= 0 ,0
Exp/Cntr=0.3,0.1

Type RM Length L Ch R = 1 ,19066.6 ,302.6,316.3,328
XS GIS Cut Line= 2
     1980711.695      199035.499     1980841.904      199247.305
#Sta/Elev= 30
       0 2375.87    13.1 2371.12    22.9 2366.63    32.7 2363.33    55.6 2357.86
    65.4 2355.89    81.8 2355.01    88.3 2354.22    91.6 2353.04    94.9 2351.22
    98.1 2350.23   101.4 2349.86     108 2349.78   114.5  2350.3     121 2351.77
   134.1 2356.84   137.4 2357.42   150.5 2357.91     157 2358.46   166.8 2360.52
   173.4  2362.5   179.9 2365.21   196.3 2370.91   199.6  2372.6   206.1 2377.13
   215.9 2381.94   225.7 2387.45     229 2388.92   242.1 2393.49   248.6 2395.45
#Mann= 3 ,-1 , 0
       0     .12       0    98.1    .045       0   114.5     .12       0
#XS Ineff= 2 , 0
           87.46 2357.74
Permanent Ineff=
       F       F
Bank Sta=98.1,114.5
XS Rating Curve= 0 ,0
Exp/Cntr=0.3,0.1

Type RM Length L Ch R = 1 ,18750.3 ,162.2,165.5,167.5
XS GIS Cut Line= 2
     1980524.195      199063.277     1980522.459      199323.694
#Sta/Elev= 30
       0  2392.1     3.3 2391.17     6.5 2389.77      13 2386.22    16.3 2384.96
      26 2382.36    29.3 2381.12    42.3 2375.15    55.3 2369.99    71.6 2361.98
    74.9 2360.12    78.1 2357.71    87.9 2348.32   90.59 2346.91    91.2 2346.59
    94.4 2346.14   104.2 2346.84   117.2 2350.61   130.2 2351.52   146.5 2350.72
   156.2 2351.07   162.8 2351.95     179  2355.5   201.8 2357.99   214.8 2358.77
   221.4 2359.58   234.4 2362.58   237.6 2363.65   250.7  2368.7   260.4 2372.94
#Mann= 3 ,-1 , 0
       0     .12       0   90.59    .045       0   104.2     .12       0
#XS Ineff= 2 , 0
                          130.03         2353.28
Permanent Ineff=
       F       F
Bank Sta=90.59,104.2
XS Rating Curve= 0 ,0
Exp/Cntr=0.3,0.1

Type RM Length L Ch R = 1 ,18584.8 ,144.3,140.8,136.4
XS GIS Cut Line= 2
     1980399.237      199090.419     1980366.684       199353.44
#Sta/Elev= 30
       0  2370.4     9.8 2367.13    19.6 2364.48    42.5 2360.29    68.7  2357.8
    81.8 2358.18    85.1 2358.08    88.3 2357.63    91.6 2356.86    98.2 2354.69
     108 2349.97   111.2 2348.96   121.1 2347.93   124.3 2347.19   130.9 2344.98
   134.2 2344.03   137.4  2343.8   140.7 2343.92   145.9 2344.87     157 2349.33
   166.9 2353.94   189.8 2359.26   199.6 2362.17   202.9 2363.32   222.5 2371.63
   225.8 2372.91     229 2373.74   245.4 2374.85   248.7 2374.54     265  2371.4
#Mann= 3 , 0 , 0
       0     .12       0   130.9    .045       0   145.9     .12       0
Bank Sta=130.9,145.9
XS Rating Curve= 0 ,0
Exp/Cntr=0.3,0.1

Type RM Length L Ch R = 1 ,18443.9 ,120,85.2,48.8
XS GIS Cut Line= 3
     1980243.941      199109.965     1980249.497       199228.44
     1980361.476      199349.534
#Sta/Elev= 30
       0 2364.35    12.8  2358.5    19.2 2356.29    35.3 2352.77    48.1 2351.72
    54.5 2350.61    57.7 2349.23    64.1 2345.46    81.2 2341.52    89.8 2341.24
    96.2 2341.58   102.6 2342.94   105.8 2344.29     109 2346.02   118.6 2352.35
   128.3 2353.88   144.5 2354.53   154.2 2355.67   157.4 2356.76   167.1 2361.46
   170.4 2362.27   189.8 2365.06   202.7  2366.4   205.9 2367.09   212.4 2369.75
   218.9 2371.24     248 2372.79   264.1 2372.54   273.8 2371.41   283.5 2371.22
#Mann= 3 , 0 , 0
       0     .12       0    81.2    .045       0    96.2     .12       0
Bank Sta=81.2,96.2
XS Rating Curve= 0 ,0
Exp/Cntr=0.3,0.1

Type RM Length L Ch R = 1 ,18358.7 ,141.3,141.6,141.8
XS GIS Cut Line= 3
     1980111.997      199255.798      1980249.15       199254.93
     1980362.865      199369.514
#Sta/Elev= 30
       0  2350.7    16.3  2352.5    29.4 2352.48    58.8 2354.03    65.3 2353.65
    71.8 2352.43    75.1 2350.54    78.4 2347.48    81.6 2342.92    84.9 2340.01
   87.17 2339.17    91.4 2338.11  101.55  2339.2   104.5 2340.32   107.8 2342.51
   120.8  2354.2   124.1 2355.05   137.2 2355.08   140.4 2355.64   153.3 2358.24
   166.2  2362.2   179.1 2364.76   201.7  2368.1   211.4 2370.15   221.1 2371.27
   240.5 2371.22   263.1 2369.43   272.8 2368.08   285.7 2367.47   298.6 2365.26
#Mann= 3 , 0 , 0
       0     .12       0   87.17    .045       0  101.55     .12       0
Bank Sta=87.17,101.55
XS Rating Curve= 0 ,0
Exp/Cntr=0.3,0.1

Type RM Length L Ch R = 1 ,18217.1 ,148.9,143.8,138.1
XS GIS Cut Line= 2
     1980105.688       199396.28     1980364.578      199396.941
#Sta/Elev= 30
       0 2319.81     3.3 2319.04     6.6  2319.5    13.1 2322.54    16.4 2323.36
    45.9 2324.13    55.7    2325      59 2324.24    68.8 2320.39    81.9 2318.86
    85.2 2317.35    98.3 2309.22   101.6  2308.5  105.91 2305.86   111.4 2304.57
   121.2 2305.89   127.8 2308.22   131.1 2311.19   137.6 2318.84   140.9 2320.54
   144.2 2321.52   147.5 2321.63     154 2320.87   160.6 2321.03   167.1 2323.54
   183.5 2331.32   203.2 2336.23   226.1 2344.44   252.3 2351.61   258.9 2353.03
#Mann= 3 , 0 , 0
       0     .12       0  105.91    .045       0   121.2     .12       0
Bank Sta=105.91,121.2
XS Rating Curve= 0 ,0
Exp/Cntr=0.3,0.1

Type RM Length L Ch R = 1 ,18073.3 ,223.2,218.2,210.5
XS GIS Cut Line= 3
     1980123.154      199558.069     1980303.709      199516.402
     1980361.001      199440.013
#Sta/Elev= 30
       0  2308.7   26.082306.154    35.8 2307.22    42.3 2307.04   60.212305.151
    61.8 2304.77      65 2303.08    74.8 2293.87   100.8 2274.23   110.5 2266.16
     117 2262.04   123.5 2258.93   126.8 2258.03     130 2257.54     143 2257.93
   146.3 2258.15   149.5 2257.77   152.8 2258.11     156 2259.24   162.5 2263.32
   165.8 2266.64   172.3 2275.89   175.6 2279.08   178.8 2280.47     198 2286.01
   217.1 2293.81   229.9 2300.35   255.3 2311.76   261.7 2315.52   280.8 2328.02
#Mann= 5 ,-1 , 0
       0    .016       0   26.08     .06       0   60.21     .12       0
   126.8    .045       0     143     .12       0
Bank Sta=126.8,143
XS Rating Curve= 0 ,0
Exp/Cntr=0.3,0.1

Type RM Length L Ch R = 1 ,17855.2 ,224.9,218.5,210.9
XS GIS Cut Line= 3
     1980204.751      199795.916     1980395.723      199686.541
     1980456.487      199571.958
#Sta/Elev= 30
       0 2291.67     9.7 2291.83   41.462289.766    45.3 2289.16    48.6  2287.6
    71.2 2268.25    77.7 2263.12    93.9 2251.76   103.6 2244.37     110 2241.08
     123 2235.77   137.5 2235.61   152.1 2235.77   165.1 2234.57   171.5 2234.89
   174.8 2235.57     178 2236.51   187.7 2240.82   207.1  2245.4   216.8 2245.82
   239.5 2244.52   249.3 2245.15   252.5 2246.16   265.5 2253.17     272 2255.24
   294.6 2268.06   301.1  2271.3   314.1 2275.84   333.6 2281.06   349.8 2287.58
#Mann= 4 ,-1 , 0
       0    .016       0   41.46     .12       0     123    .045       0
   137.5     .12       0
Bank Sta=123,137.5
XS Rating Curve= 0 ,0
Exp/Cntr=0.3,0.1

Type RM Length L Ch R = 1 ,17636.7 ,199.5,206.8,213.2
XS GIS Cut Line= 4
     1980333.223      199948.694     1980439.126      199912.236
     1980517.251      199827.166     1980616.209      199795.916
#Sta/Elev= 30
       0 2274.77     9.6 2266.71    22.4  2257.8    35.2 2249.82    44.8 2246.11
    57.6 2242.12    83.2 2235.35      96 2233.59     112 2232.44   118.4 2232.64
   134.5 2229.48   145.82225.055   150.5 2224.64   160.1 2225.12   166.5 2226.24
     173 2226.51   179.4 2225.09   185.8 2222.32     189 2222.51   195.4 2225.89
   201.8 2227.85   214.7 2228.76   221.1 2230.72   230.8 2232.42   243.7 2237.87
   256.7 2246.22   272.9 2258.02   282.6 2262.52   295.6 2271.12   331.3 2290.72
#Mann= 3 ,-1 , 0
       0     .12       0   145.8    .045       0   160.1     .12       0
Bank Sta=145.8,160.1
XS Rating Curve= 0 ,0
Exp/Cntr=0.3,0.1

Type RM Length L Ch R = 1 ,17429.8 ,239.7,225,209
XS GIS Cut Line= 3
     1980458.655      200118.745     1980665.807      199999.011
     1980703.015      199927.861
#Sta/Elev= 30
       0 2254.68    16.4  2249.3    42.6 2239.93    45.9 2238.53    68.8 2226.29
    75.4 2223.81    81.9    2222    88.5 2221.04     118 2217.76   124.6 2215.82
   131.1  2212.9   137.7 2210.59   144.2 2209.56   151.1 2210.54   160.6 2212.28
   173.7 2215.78   183.6 2219.26   190.1 2220.83   193.4 2222.35   219.6  2239.3
   229.4 2247.05   232.7 2250.17     236 2254.32   239.3  2256.3   252.1 2261.02
   261.8 2263.57   277.8  2268.6   290.6 2273.92   313.1 2280.74   319.6 2282.07
#Mann= 3 ,-1 , 0
       0     .12       0   137.7    .045       0   151.1     .12       0
Bank Sta=137.7,151.1
XS Rating Curve= 0 ,0
Exp/Cntr=0.3,0.1

Type RM Length L Ch R = 1 ,17204.8 ,295.2,286,275.4
XS GIS Cut Line= 3
     1980694.334      200332.374     1980770.723       200137.93
     1980784.612      200014.666
#Sta/Elev= 30
       0 2260.99     9.8  2255.8    22.8 2246.38    26.1  2245.6   33.57 2247.27
    58.8 2245.05      62 2243.98   66.882241.033    78.3 2232.07   101.2 2217.22
   117.5 2208.14     124  2205.3   133.8 2202.03   146.9 2201.06   156.7 2200.62
   161.72201.075     173 2203.33   182.8 2207.74   186.1 2208.71   189.3 2208.93
   208.9 2207.35   215.4 2208.43   218.7 2209.56     235 2217.51   261.1 2228.57
   277.5 2236.43   290.5 2240.82   310.1 2250.59   326.4 2257.75     333 2260.08
#Mann= 5 ,-1 , 0
       0     .12       0   33.57    .016       0   66.88     .12       0
   146.9    .045       0   161.7     .12       0
Bank Sta=146.9,161.7
XS Rating Curve= 0 ,0
Exp/Cntr=0.3,0.1

Type RM Length L Ch R = 1 ,16918.8 ,347.5,366.7,383.6
XS GIS Cut Line= 2
     1981027.668      200332.374     1981010.307       200044.18
#Sta/Elev= 30
       0 2228.63    16.2 2229.63   25.742229.284    32.4 2228.01    35.7 2226.72
    38.9  2224.8    42.2 2222.49    58.4 2209.67    74.6 2198.26    81.1 2194.14
    90.8 2189.06    97.3 2186.87   116.8 2184.48   129.8 2180.05   136.2 2178.62
     146 2178.22   152.5 2178.75   162.2 2179.73   168.7 2182.19   171.9 2184.75
   175.2 2189.15   184.9 2205.64   194.6 2220.61   197.9 2224.27   201.1 2226.34
   230.3 2242.93   256.3 2256.48     266 2262.11   285.5  2274.3   288.7 2275.91
#Mann= 4 ,-1 , 0
       0    .016       0   25.74     .12       0   136.2    .045       0
   152.5     .12       0
Bank Sta=136.2,152.5
XS Rating Curve= 0 ,0
Exp/Cntr=0.3,0.1

Type RM Length L Ch R = 1 ,16552.1 ,285.3,286.4,285.5
XS GIS Cut Line= 3
     1981256.834       200387.93     1981366.209      200261.194
     1981393.987      200130.986
#Sta/Elev= 30
       0 2211.36     3.2 2209.31    6.05 2208.41    38.6 2209.36    45.1 2207.69
   51.262204.118   58.332199.286    64.4 2194.54    70.8 2188.18    90.1 2173.76
    96.6 2167.99   106.2 2163.42   125.6 2160.16   135.2 2159.82  140.022160.164
   141.6  2160.5   144.9 2162.54   148.1 2165.74   151.3 2167.12     161 2168.86
   167.4  2171.4   177.2 2176.36   183.6 2180.61   196.6 2188.08   203.1 2193.27
   209.6 2197.29   219.4 2201.84   229.1    2205   242.1 2210.64   300.5 2238.26
#Mann= 6 ,-1 , 0
       0     .06       0    6.05    .016       0   51.26     .08       0
   58.33     .12       0   125.6    .045       0  140.02     .12       0
Bank Sta=125.6,140.02
XS Rating Curve= 0 ,0
Exp/Cntr=0.3,0.1

Type RM Length L Ch R = 1 ,16265.7 ,344.7,354.7,362.9
XS GIS Cut Line= 2
     1981492.945      200523.347     1981670.029      200323.694
#Sta/Elev= 30
       0 2186.96    3.132187.175    22.8 2188.76   27.562187.662    32.6 2184.82
    45.6 2175.09    52.1 2170.98    78.1 2159.12    87.9 2155.51   100.9 2153.88
   107.4 2152.25   113.9 2149.76   120.4 2146.66   133.4 2143.64   146.4 2142.53
   149.72143.338   159.5 2148.95     166 2151.88   169.2 2154.53   182.2 2167.46
   188.8 2173.29   195.3 2179.67   208.3 2193.01   211.5  2195.9   221.3 2203.48
   224.6 2206.83   231.1  2214.9   247.3 2228.26   257.1 2236.93   266.9 2243.84
#Mann= 5 ,-1 , 0
       0     .06       0    3.13    .016       0   27.56     .12       0
   133.4    .045       0   149.7     .12       0
Bank Sta=133.4,149.7
XS Rating Curve= 0 ,0
Exp/Cntr=0.3,0.1

Type RM Length L Ch R = 1 ,15911   ,303.2,300.5,296.6
XS GIS Cut Line= 3
     1981628.362      200785.499     1981814.126      200696.958
     1981920.029      200686.541
#Sta/Elev= 30
       0 2202.37     6.5 2197.82     9.8 2194.91    13.1 2190.45    18.22180.073
    22.9 2171.09    26.1 2167.04    29.4  2164.7    32.7 2163.64    58.8 2163.94
    66.92162.478    71.9 2160.11    75.1 2157.85    88.2 2147.26   107.8 2132.52
   111.1 2130.81   124.1  2127.7   133.9  2127.1   140.5 2127.45     147 2130.15
   156.8 2135.35   169.9 2139.27   189.4 2142.74   218.7 2145.02   228.4 2147.68
   254.2 2159.37   263.8 2164.65     280 2176.48   289.6 2181.78   312.2  2196.6
#Mann= 5 ,-1 , 0
       0     .06       0    18.2    .016       0    66.9     .12       0
   124.1    .045       0   140.5     .12       0
Bank Sta=124.1,140.5
XS Rating Curve= 0 ,0
Exp/Cntr=0.3,0.1

Type RM Length L Ch R = 1 ,15610.5 ,305.9,303.6,300.4
XS GIS Cut Line= 2
     1981772.459      201068.486     1982020.723      200901.819
#Sta/Elev= 30
       0 2149.46      13  2148.9   19.192148.078    32.5 2146.56    35.8  2145.7
    42.2 2142.37    45.5 2142.04      52 2143.12    58.5 2143.15    71.5 2142.34
    87.8 2140.36    94.3 2137.91   108.22128.062     117 2122.98   123.5 2120.78
     130 2119.51   136.5 2118.79   146.3 2119.46   152.8 2122.17   162.5 2127.86
   172.3 2132.51   201.5    2148   214.5 2156.96   224.3 2162.16     234 2167.99
   240.5 2174.07   256.8 2185.21   269.8 2192.74   279.5 2199.34     299 2208.88
#Mann= 5 ,-1 , 0
       0     .12       0   19.19    .016       0   108.2     .12       0
     130    .045       0   146.3     .12       0
Bank Sta=130,146.3
XS Rating Curve= 0 ,0
Exp/Cntr=0.3,0.1

Type RM Length L Ch R = 1 ,15307   ,439.3,436,431.1
XS GIS Cut Line= 2
     1981998.154      201280.291     1982209.959      201096.263
#Sta/Elev= 30
       0 2120.81     3.3 2122.72     6.5 2123.77   11.052123.984    26.1 2123.38
    35.9 2122.28    42.4 2122.67   47.332121.999    68.5 2118.91    91.4 2117.07
   104.4 2117.55   110.9 2117.08   120.7  2114.9   130.5 2111.11   145.4 2107.69
   153.3 2107.04   160.72107.702   166.4 2110.77     186 2131.65   189.2 2136.14
   192.5 2141.95     199 2155.17   202.3 2161.13   205.5 2165.36   208.8 2168.11
   221.9 2175.87   234.9 2187.15   238.2 2189.49   267.5 2206.94   280.6 2213.28
#Mann= 5 ,-1 , 0
       0     .12       0   11.05    .016       0   47.33     .12       0
   145.4    .045       0   160.7     .12       0
Bank Sta=145.4,160.7
XS Rating Curve= 0 ,0
Exp/Cntr=0.3,0.1

Type RM Length L Ch R = 1 ,14870.9 ,304.3,304,302.7
XS GIS Cut Line= 2
      1982312.39      201549.388     1982492.945      201330.638
#Sta/Elev= 30
       0 2115.79     3.3 2113.64   13.732103.873    16.3  2102.3    19.6 2101.48
    39.1 2101.43    48.9 2100.65   55.162102.527    61.9 2104.63    68.5 2104.17
    97.8 2097.83   110.8 2092.35   117.4 2090.37   140.2 2088.43   153.2 2088.29
   156.5 2088.32   159.8 2090.52     163 2097.58   166.3 2106.02   169.5  2112.4
   172.8 2117.06   179.3 2123.89   185.8 2129.48   198.9 2139.34   228.2 2167.52
   234.7 2172.97   247.8 2181.68   257.6 2190.38   267.3 2200.08   283.6 2212.87
#Mann= 5 ,-1 , 0
       0     .12       0   13.73    .016       0   55.16     .12       0
   140.2    .045       0   156.5     .12       0
Bank Sta=140.2,156.5
XS Rating Curve= 0 ,0
Exp/Cntr=0.3,0.1

Type RM Length L Ch R = 1 ,14567   ,295.4,295.3,295.2
XS GIS Cut Line= 2
     1982546.765       201731.68     1982723.848      201502.513
#Sta/Elev= 30
       0 2085.75   15.812085.913    22.8 2086.82      39 2086.98    52.1 2085.91
    55.3 2085.06   57.222084.077    58.6 2083.37    65.1 2076.99    68.3 2075.11
    74.8 2074.14    87.9 2073.63    91.1    2074    97.6  2078.2   104.1 2081.82
   136.7 2096.33   143.2 2099.96   152.9 2106.86   159.4 2110.32   169.2 2116.85
   175.7 2121.65   185.5 2127.49   195.2 2134.51   214.8 2147.54   224.5  2155.2
   227.8 2157.17   237.6 2161.82   263.6 2178.95   279.8 2188.66   289.6 2195.07
#Mann= 5 ,-1 , 0
       0     .12       0   15.81    .016       0   57.22     .12       0
    74.8    .045       0    91.1     .12       0
Bank Sta=74.8,91.1
XS Rating Curve= 0 ,0
Exp/Cntr=0.3,0.1

Type RM Length L Ch R = 1 ,14271.7 ,301.1,301.9,301.8
XS GIS Cut Line= 2
      1982789.82      201900.083     1982958.223      201679.597
#Sta/Elev= 30
       0 2072.56     1.62072.662    13.1  2073.5    26.1  2073.6    35.9 2073.14
    39.2 2072.57   43.012071.212    52.2 2066.37    55.5 2065.16    58.8  2064.2
    65.3 2063.56    75.1 2062.76    81.6 2063.58    84.9 2064.44   107.7 2073.67
   117.5 2079.43   130.6 2086.06   143.6 2094.88   150.1 2100.13   163.2 2109.78
   169.7 2115.74   176.3  2121.1     186 2130.54   189.3 2133.43   202.4 2142.27
   208.9 2148.54   231.8 2166.65   248.1 2180.25   267.6 2194.92   277.4  2203.7
#Mann= 5 ,-1 , 0
       0     .12       0     1.6    .016       0   43.01     .12       0
    65.3    .045       0    81.6     .12       0
Bank Sta=65.3,81.6
XS Rating Curve= 0 ,0
Exp/Cntr=0.3,0.1

Type RM Length L Ch R = 1 ,13969.7 ,402.4,406.3,408
XS GIS Cut Line= 2
     1983017.251      202073.694     1983185.654       201856.68
#Sta/Elev= 30
       0 2063.24     6.5 2062.07      36 2062.29    39.2 2061.63   42.442059.696
      49 2054.56    55.2 2052.96    62.1 2052.62    70.2 2053.04    78.5 2053.81
      85 2055.71    88.3 2055.97    98.1 2054.99   101.4 2055.51   104.6 2056.78
   107.9 2058.86   114.4  2069.9   117.7 2073.31   137.3 2087.39   150.4 2099.22
   160.2 2104.67   163.5 2107.03     170 2115.29   176.6 2122.34   179.9 2125.29
   196.2 2137.81   222.4 2156.46   238.7 2171.93   261.6 2188.54   274.7 2197.07
#Mann= 4 ,-1 , 0
       0    .016       0   42.44     .12       0    55.2    .045       0
    70.2     .12       0
Bank Sta=55.2,70.2
XS Rating Curve= 0 ,0
Exp/Cntr=0.3,0.1

Type RM Length L Ch R = 1 ,13563.4 ,282.8,282.9,282.4
XS GIS Cut Line= 2
     1983253.362      202320.222     1983459.959      202103.208
#Sta/Elev= 30
       0  2092.8    19.5 2077.82    22.8 2072.76    29.3 2061.42   36.482054.397
    39.1 2052.46    42.3 2051.33    68.4 2052.73    71.6 2052.06   75.382049.997
    91.2 2038.32    97.7 2036.15     101 2036.04     114 2036.24   117.2 2036.84
   120.5 2039.11   123.8 2042.97     127 2045.69   130.3 2048.13   133.5 2048.95
   146.6 2050.16   172.6 2050.45   185.6 2053.67   192.2 2056.67   201.9 2062.51
   221.5 2071.64     254 2084.18   276.8 2094.27   289.9 2098.95   299.6 2101.58
#Mann= 5 ,-1 , 0
       0     .12       0   36.48    .016       0   75.38     .12       0
    97.7    .045       0     114     .12       0
Bank Sta=97.7,114
XS Rating Curve= 0 ,0
Exp/Cntr=0.3,0.1

Type RM Length L Ch R = 1 ,13280.5 ,303.8,301.5,298.5
XS GIS Cut Line= 3
     1983444.334      202528.555     1983555.445      202410.499
     1983675.237      202349.736
#Sta/Elev= 30
       0 2055.91     3.2 2054.88    16.2 2053.25    19.4 2051.95    32.4 2044.84
    35.7 2043.78      382043.816    48.6  2044.5    68.1 2043.35    74.6 2040.34
   82.032035.502      94 2028.02   98.942026.201   103.8 2025.37   110.2 2025.24
  115.082026.313   129.7 2034.02   139.4 2037.17   162.1 2048.25   181.8 2056.71
   188.3 2060.53   198.2 2067.75   201.4 2070.87   204.7 2074.84   211.3 2084.01
   217.8 2090.17   234.2 2101.93   250.6 2114.33   273.5 2129.78   296.4 2147.69
#Mann= 5 ,-1 , 0
       0     .12       0      38    .016       0   82.03     .12       0
   98.94    .045       0  115.08     .12       0
Bank Sta=98.94,115.08
XS Rating Curve= 0 ,0
Exp/Cntr=0.3,0.1

Type RM Length L Ch R = 1 ,12979   ,271.7,267.9,263.3
XS GIS Cut Line= 3
     1983663.084      202747.305     1983751.626      202627.513
     1983796.765      202495.569
#Sta/Elev= 30
       0 2056.45    16.2 2045.91   26.592035.848    29.1 2033.55    32.4 2031.94
    61.5 2029.81      68 2028.81    71.2 2027.32   76.832023.209      81 2020.67
   86.282018.905    93.9  2018.5  102.022018.751   106.9 2019.69   110.1 2022.54
   116.6 2030.45   119.8 2032.18   129.5 2035.43   139.2 2035.56     149 2037.83
   158.7 2041.64   168.4 2047.96   184.6 2054.23   197.6 2057.67   207.3 2061.59
   223.6 2069.65   233.3 2075.68   265.7 2099.18   272.2 2103.24   288.4 2115.61
#Mann= 5 ,-1 , 0
       0     .12       0   26.59    .016       0   76.83     .12       0
   86.28    .045       0  102.02     .12       0
Bank Sta=86.28,102.02
XS Rating Curve= 0 ,0
Exp/Cntr=0.3,0.1

Type RM Length L Ch R = 1 ,12711.1 ,259.6,257.1,254.5
XS GIS Cut Line= 2
     1983913.084      202877.513      1984031.14      202632.722
#Sta/Elev= 30
       0 2023.69     3.3 2023.18    6.912021.497    13.1 2020.18   49.022017.953
    58.9 2017.55    65.5 2016.54    68.8 2015.33    75.3  2011.1    78.6  2009.8
    81.9 2009.63    91.7 2011.64      95 2011.79   100.6 2010.42   115.6 2010.27
   117.9 2010.89   121.2 2013.82   127.7 2022.86     131 2026.65   134.2 2028.63
   140.8  2031.1   153.9 2041.05   186.6 2070.14   199.7 2080.82   206.3 2086.94
   216.1 2095.06   235.8 2105.92   245.6 2115.35     262 2126.86   271.8 2136.27
#Mann= 5 ,-1 , 0
       0     .12       0    6.91    .016       0   49.02     .12       0
   100.6    .045       0   115.6     .12       0
Bank Sta=100.6,115.6
XS Rating Curve= 0 ,0
Exp/Cntr=0.3,0.1

Type RM Length L Ch R = 1 ,12454   ,309.5,298.3,287.1
XS GIS Cut Line= 3
      1984156.14      202979.944     1984197.807      202860.152
     1984206.487      202726.472
#Sta/Elev= 30
       0 2029.15     9.8 2022.68    16.3 2017.16    19.5 2014.98   21.052014.689
    22.8 2014.36    29.3 2014.99      39 2014.46      52 2013.59   56.012012.481
    58.5 2011.08      65    2004    68.3 2001.26    71.6 1999.32   73.821998.786
    81.3 1998.33    87.8 1998.48    91.1 1999.08    94.3 2001.45   113.8 2019.14
   120.3 2024.29   123.6 2026.25   139.9 2032.17   149.7 2036.33   192.2 2054.87
   228.1 2071.53   231.4  2073.2   237.9 2077.87   244.5 2081.96   260.8 2094.55
#Mann= 5 ,-1 , 0
       0     .12       0   21.05    .016       0   56.01     .12       0
   73.82    .045       0    87.8     .12       0
Bank Sta=73.82,87.8
XS Rating Curve= 0 ,0
Exp/Cntr=0.3,0.1

Type RM Length L Ch R = 1 ,12155.7 ,267,275.1,282.4
XS GIS Cut Line= 2
     1984492.945      203014.666     1984447.807      202736.888
#Sta/Elev= 30
       0 2012.12   14.312012.577    45.8 2012.86    62.2 2011.93    65.4  2010.3
    81.8 1996.23    85.1 1993.69   87.641992.558    91.6 1991.82   101.4 1992.27
     108 1992.85   117.8 1992.23   124.4 1995.11   134.2 1996.53   137.4 1997.58
   150.5 2004.31   173.4  2014.4   186.5 2022.21   199.6 2032.03   202.9 2033.96
   209.4  2036.7   219.2  2042.9   232.3 2053.94   242.2 2061.35   248.7  2064.7
   265.1 2078.24   268.3 2080.67   274.9 2084.43   278.2 2086.87   281.4 2090.04
#Mann= 4 ,-1 , 0
       0    .016       0   14.31     .12       0   87.64    .045       0
   101.4     .12       0
#XS Ineff= 2 , 0
                           125.7         1999.05
Permanent Ineff=
       F       F
Bank Sta=87.64,101.4
XS Rating Curve= 0 ,0
Exp/Cntr=0.3,0.1

Type RM Length L Ch R = 1 ,11880.7 ,281.6,305.3,328.2
XS GIS Cut Line= 3
      1984633.57      203011.194     1984730.793      202917.444
     1984763.779      202733.416
#Sta/Elev= 30
       0 2012.23    16.1 2011.64    25.7  2011.8    51.4 2010.83    80.4 2008.96
    99.7 2001.48   106.1 2000.41   125.4 1998.46   131.8 1997.26   144.9 1995.67
   151.5 1994.29   167.9 1988.48     181 1982.03  189.271980.186   194.1 1979.93
   203.9 1980.07   210.5 1980.68   220.3  1983.2   226.9 1986.22   233.5 1988.68
   243.3  1993.6   249.9  1996.2   253.1 1998.21     263 2005.55   266.3 2008.57
   272.8 2015.29   285.9 2029.68   289.2  2032.9   308.9 2049.97     322 2062.46
#Mann= 3 ,-1 , 0
       0     .12       0  189.27    .045       0   203.9     .12       0
Bank Sta=189.27,203.9
XS Rating Curve= 0 ,0
Exp/Cntr=0.3,0.1

Type RM Length L Ch R = 1 ,11575.4 ,359.2,337.9,315.3
XS GIS Cut Line= 3
     1984822.807      203094.527      1985008.57      203023.347
     1985064.126      202907.027
#Sta/Elev= 30
       0 1998.29   29.131995.823    81.5 1992.63    94.6 1990.93   101.1 1988.37
   104.4  1986.7   107.6 1984.65   114.1 1979.78   120.7 1973.84   123.9 1971.81
   128.7 1970.67   130.4 1970.41   143.5 1970.65     150 1971.22   156.5  1972.8
   172.8 1974.33   179.4 1974.45   185.9 1973.76   202.2 1974.12   224.7 1972.76
   231.2 1972.92   237.6 1973.96   247.3 1977.95   256.9 1984.85   263.4 1988.89
   292.4 2004.68   298.8 2007.77   308.5 2013.75     315 2016.91   327.8 2024.33
#Mann= 4 ,-1 , 0
       0    .016       0   29.13     .12       0   128.7    .045       0
   143.5     .12       0
Bank Sta=128.7,143.5
XS Rating Curve= 0 ,0
Exp/Cntr=0.3,0.1

Type RM Length L Ch R = 1 ,11237.5 ,297.5,289.6,281.2
XS GIS Cut Line= 2
     1985236.001      203247.305     1985303.709       202981.68
#Sta/Elev= 30
       0  1962.8    16.3 1963.62    19.6 1964.42    29.4 1969.81    32.6 1970.76
   36.661970.938    52.2 1971.44    65.3 1970.89    68.5  1970.3   71.561968.612
    75.1 1965.51    84.8  1955.7    88.1 1954.22    97.9 1953.87   101.2 1954.13
   104.4  1955.6     111 1960.61     124  1972.8   130.5 1976.95   137.1 1979.42
   146.8 1982.01   163.2 1985.39   179.5 1989.79   192.5  1994.5   212.1 2002.69
   221.9 2005.49     235  2010.2   257.8 2020.93   270.9 2030.18   274.1 2031.83
#Mann= 5 ,-1 , 0
       0     .12       0   36.66    .016       0   71.56     .12       0
    88.1    .045       0   101.2     .12       0
Bank Sta=88.1,101.2
XS Rating Curve= 0 ,0
Exp/Cntr=0.3,0.1

Type RM Length L Ch R = 1 ,10947.9 ,299.1,329.8,359.2
XS GIS Cut Line= 2
     1985557.182      203297.652     1985524.195      203007.722
#Sta/Elev= 30
       0 1958.36     6.6  1953.9     9.8 1952.32   11.331952.037    13.1 1951.71
    32.8 1953.16   46.681953.395    88.5  1949.8    91.8 1948.49    95.1 1946.78
   97.071946.339   101.6    1946   111.5  1946.2   114.8 1946.74   121.3 1948.74
   124.6 1949.28     141 1949.33   157.4 1948.63   170.5  1947.6   173.8 1947.84
     177  1948.9   180.3 1951.31   186.9 1957.32   193.4 1961.98   226.2 1981.78
   236.1 1988.55   245.9 1994.63   252.5  1999.1   278.7 2018.02   291.8 2028.16
#Mann= 5 ,-1 , 0
       0     .12       0   11.33    .016       0   46.68     .12       0
   97.07    .045       0   111.5     .12       0
#XS Ineff= 2 , 0
           88.85 1952.67
Permanent Ineff=
       F       F
Bank Sta=97.07,111.5
XS Rating Curve= 0 ,0
Exp/Cntr=0.3,0.1
